--- KeeneyCrk.prj (project) ---

Proj Title=KeeneyCrk
Current Plan=p01
Default Exp/Contr=0,0
English Units
Geom File=g01
Flow File=f01
Plan File=p01
BEGIN DESCRIPTION:
END DESCRIPTION:
DSS Export Rating Curves= 0
DSS Export Rating Curve Sorted= 0
DSS Export Volume Flow Curves= 0
DXF OffsetX= 0
DXF OffsetY= 0
DXF ScaleX= 0
DXF ScaleY= 0

--- KeeneyCrk.p01 (plan) ---

Plan Title=Floodplain
Program Version=4.00
Geom File=g01
Flow File=f01
K Sum by GR=0
Std Step Tol=0.01
Critical Tol=0.01
Num of Std Step Trials=20
Max Error Tol=0.3
Flow Tol Ratio=0.001
Split Flow NTrial=30
Split Flow Tol=0.02
Split Flow Ratio=0.02
Log Output Level=0
Friction Slope Method=1
Unsteady Friction Slope Method=2
Unsteady Bridges Friction Slope Method=1
Global Log Level=0
CheckData=False
Run HTab=0
Run UNet=0
Run PostProcess=0
UNET Theta=0
UNET Theta Warmup=0
UNET ZTol=0
UNET ZSATol=0
UNET MxIter=0
UNET MaxInSteps=0
UNET DtIC=0
UNET DtMin=0
UNET MaxCRTS=0
UNET WFStab=0
UNET SFStab=0
UNET WFX=0
UNET SFX=0
UNET DSS MLevel=0
UNET DZMax Abort=0
UNET Convert EG Bridges=0
UNET Use Existing IB Tables=0
UNET Froude Limit=0
UNET Froude Power=0
Write IC File=0
Echo Input=False
Echo Output=False
Write Detailed=0

--- KeeneyCrk.f01 (steady flow) ---

Flow Title=NFF Regression Equation
Program Version=4.00
Number of Profiles=1
Profile Names=P100yr
River Rch & RM=KeeneyCrk,Main      ,21977.9
546.8267
River Rch & RM=KeeneyCrk,Main      ,19577.9
582.1193
River Rch & RM=KeeneyCrk,Main      ,19292.6
650.2291
River Rch & RM=KeeneyCrk,Main      ,18077.9
660.3861
River Rch & RM=KeeneyCrk,Main      ,17837.3
812.2956
River Rch & RM=KeeneyCrk,Main      ,15651.2
864.4113
River Rch & RM=KeeneyCrk,Main      ,15391.4
963.4635
River Rch & RM=KeeneyCrk,Main      ,13294.6
1021.841
River Rch & RM=KeeneyCrk,Main      ,12178
1134.597
River Rch & RM=KeeneyCrk,Main      ,9976.6
1166.504
River Rch & RM=KeeneyCrk,Main      ,7169.1
1292.921
River Rch & RM=KeeneyCrk,Main      ,6658.3
1519.864
River Rch & RM=KeeneyCrk,Main      ,4869.5
1590.264
Boundary for River Rch & Prof#=KeeneyCrk,Main      ,1
Up Type=0
Dn Type=3
Dn Slope=0.1284

--- KeeneyCrk.g01 (geometry) ---

Geom Title=USGS 3m DEM
Program Version=4.10

River Reach=KeeneyCrk       ,Main
Reach XY= 30
     1972299.095      385548.768     1971667.151      384769.254
     1971573.401      384338.699      1971649.79      383968.907
     1972052.035      383543.722     1971951.873      382982.796
     1972073.401      382505.366     1971918.887       382137.31
     1970927.213      381501.991     1970714.524      380784.155
     1970800.831      380552.241     1970418.887      380312.657
     1970229.651      379751.893     1969417.834      378914.036
     1969248.748      378461.963     1968667.651      377907.353
     1968406.734      377939.393     1967398.053      377078.282
     1966784.425      376835.368     1966543.325      376422.914
     1965935.686      376209.372     1965092.975      376280.862
     1964881.867      376719.788     1964697.839      376752.774
     1964102.353      375349.997     1963614.506      375096.524
     1962962.924      375403.202     1961602.353        376455.9
     1960289.853      377096.524     1959516.896      377166.105

Type RM Length L Ch R = 1 ,21977.9 ,292.3,300,308.8
XS GIS Cut Line= 3
     1972561.304      385069.746     1972290.413      385543.807
     1972019.521      386017.868
#Sta/Elev= 30
       0 2159.42    19.8 2156.39    29.8 2154.28    49.6 2148.76     129 2125.13
   148.9 2120.01   248.2 2098.52     268 2095.27   317.7  2088.4   357.4 2082.16
   426.9 2074.36   526.2  2060.7   538.5 2059.39     546 2059.11   553.5 2059.26
   595.6 2060.24   625.4 2061.36     675 2063.91   694.9 2065.42   714.8 2068.29
   744.6 2074.98   764.4 2080.27   784.2 2086.13     953 2141.79     963 2143.71
   972.9  2144.8  1042.4 2146.49  1062.2 2147.74  1072.2 2149.23    1092 2154.69
#Mann= 3 , 0 , 0
       0      .1       0   538.5    .045       0   553.5      .1       0
Bank Sta=538.5,553.5
XS Rating Curve= 0 ,0
Exp/Cntr=0.3,0.1

Type RM Length L Ch R = 1 ,21677.9 ,294,300,302.7
XS GIS Cut Line= 3
     1972471.154       385003.16     1972056.058      385360.926
     1971624.876      385695.312
#Sta/Elev= 30
       0 2157.82    79.7 2154.03    89.7 2152.75    99.6 2150.47   139.5 2137.48
     259 2092.17     279 2086.03   318.8 2080.51   428.4 2068.25   540.5  2054.2
     548 2054.01   555.5 2054.63   587.7 2060.18     667 2072.24   686.9 2076.43
   716.6 2084.57   736.5 2091.26   746.4 2095.36   766.3 2106.37     796 2126.58
   805.9  2131.5   815.9 2134.26   895.2 2138.47   905.2 2139.91   915.1 2142.59
   944.8 2153.28   974.6 2162.56   994.4 2170.33  1034.1 2188.37  1093.6 2217.43
#Mann= 3 , 0 , 0
       0      .1       0   540.5    .045       0   555.5      .1       0
Bank Sta=540.5,555.5
XS Rating Curve= 0 ,0
Exp/Cntr=0.3,0.1

Type RM Length L Ch R = 1 ,21377.9 ,301.8,299.8,297.6
XS GIS Cut Line= 3
     1972393.833      384871.494     1971900.997      385105.274
     1971429.471      385386.432
#Sta/Elev= 30
       0 2154.26    59.5 2153.78     119 2151.12   148.8  2149.2   158.7 2147.07
   168.6 2143.81   307.4 2091.28   347.1 2076.68     357 2073.72     367 2071.85
   505.8 2052.06     538 2048.63     553 2047.26   555.4 2047.07   565.4 2047.33
   575.4 2049.74   635.3 2075.88   665.2 2088.09   685.2 2095.39   705.2 2101.23
   715.2 2103.31   725.1 2104.26   735.1 2104.01     785 2101.15     795 2101.65
     805 2104.17   874.9  2129.4   954.7 2159.66   994.6 2175.47  1094.5 2216.15
#Mann= 3 , 0 , 0
       0      .1       0     538    .045       0     553      .1       0
Bank Sta=538,553
XS Rating Curve= 0 ,0
Exp/Cntr=0.3,0.1

Type RM Length L Ch R = 1 ,21077.9 ,291.4,300,311.2
XS GIS Cut Line= 3
     1972207.666      384583.423      1971735.01       384858.01
     1971292.858      385184.088
#Sta/Elev= 30
       0 2160.16    49.7 2160.44    79.5 2159.74   109.3 2157.52   149.1 2152.46
     159 2150.24     169 2146.86   188.8 2138.86   208.7 2130.02   288.2  2091.7
   298.2 2087.42     318 2080.56   367.7 2067.28   539.1 2039.71   546.6 2039.26
   554.1 2039.86   606.6 2052.69   616.6 2056.16   686.5 2087.84   696.5 2092.01
   706.4 2094.79   716.4  2095.7   776.4 2097.68   796.4 2099.33   806.3 2101.63
   876.3 2123.08   926.2 2140.72   976.2 2160.59  1056.1 2195.65    1096 2215.06
#Mann= 3 , 0 , 0
       0      .1       0   539.1    .045       0   554.1      .1       0
Bank Sta=539.1,554.1
XS Rating Curve= 0 ,0
Exp/Cntr=0.3,0.1

Type RM Length L Ch R = 1 ,20777.9 ,295.2,299.9,302.5
XS GIS Cut Line= 3
     1972179.057       384501.01       1971637.7      384584.107
     1971096.869      384660.293
#Sta/Elev= 30
       0 2158.53    49.8 2160.05    79.7 2159.88    89.6 2158.54   139.4 2148.55
   159.3 2142.67   209.1 2124.37   258.9 2107.41   338.6 2081.09   388.4 2065.34
     488 2044.39   527.8  2035.1   540.2 2032.91   547.7 2032.49   555.2 2032.87
   637.1 2039.05     647 2040.34   676.8 2046.09   746.3 2061.53   756.2 2065.06
     796 2081.48   845.6  2099.4   855.5 2101.36   865.5 2102.17   905.2 2104.13
   915.1 2106.57   964.8  2126.2  1014.4  2148.4  1044.2 2161.02  1093.9 2180.59
#Mann= 3 , 0 , 0
       0      .1       0   540.2    .045       0   555.2      .1       0
Bank Sta=540.2,555.2
XS Rating Curve= 0 ,0
Exp/Cntr=0.3,0.1

Type RM Length L Ch R = 1 ,20477.9 ,291.8,300,311.6
XS GIS Cut Line= 3
     1972152.228      384326.293     1971573.227      384294.256
     1971033.318      384307.762
#Sta/Elev= 30
       0 2161.29      50    2161     160  2152.2     180 2149.22     200 2142.61
     260 2118.84   309.9 2100.44   389.9 2074.12   449.9 2057.95   572.4 2030.72
   587.4  2029.5   589.9 2029.49   599.9 2031.53   609.9 2035.78   629.9 2046.99
   639.9 2051.22   649.9 2053.54   679.9 2059.31   699.9 2061.34   799.9 2065.48
   809.9 2066.65   829.9 2073.14   909.9 2106.81   919.9 2109.37   929.9 2109.37
   949.9 2105.92   959.9 2106.58   969.9 2110.23    1060 2151.09    1120 2180.68
#Mann= 3 , 0 , 0
       0      .1       0   572.4    .045       0   587.4      .1       0
Bank Sta=572.4,587.4
XS Rating Curve= 0 ,0
Exp/Cntr=0.3,0.1

Type RM Length L Ch R = 1 ,20177.9 ,291.8,300,304.7
XS GIS Cut Line= 3
     1972170.563      384242.222     1971630.573       384004.72
     1971156.288      383750.225
#Sta/Elev= 30
       0 2162.72      40 2162.06     140 2154.19     160 2151.54     170 2148.34
     190 2138.86     270 2104.73     300 2094.24     330 2084.97   459.9  2051.7
   582.4 2025.94   597.4  2025.2   739.4 2032.67   749.4 2033.72   759.4 2036.01
   819.2 2057.72   839.1 2066.59     859  2078.3     869 2085.18   888.9 2100.35
   898.9 2106.71   908.9 2109.72   918.8 2110.31   958.7  2110.2   968.7 2110.87
   978.6 2113.79  1038.4 2145.29  1058.4 2154.44  1088.3 2166.24  1128.2 2180.09
#Mann= 3 , 0 , 0
       0      .1       0   582.4    .045       0   597.4      .1       0
Bank Sta=582.4,597.4
XS Rating Curve= 0 ,0
Exp/Cntr=0.3,0.1

Type RM Length L Ch R = 1 ,19877.9 ,308.1,300,292.3
XS GIS Cut Line= 3
     1972223.318      384173.079     1971826.284      383780.906
      1971408.78       383426.83
#Sta/Elev= 30
       0 2164.28    49.8 2164.48   139.5 2157.65   159.4 2154.29   179.4 2146.23
   199.3 2136.39   239.2 2112.28   259.1 2103.66     289 2092.93   448.4 2041.29
   518.2 2026.74   538.1 2021.58   550.6 2019.84   558.1 2019.55   565.6 2019.84
   607.8 2022.46   647.6 2026.71   667.6 2030.27   687.5 2036.29   737.2 2055.38
   767.1 2070.02   796.9  2082.1   846.7 2105.19   926.3 2139.12   936.3 2141.43
   946.2 2142.27  1035.8 2143.26  1045.8 2145.19  1055.7 2148.53  1105.5 2168.51
#Mann= 3 , 0 , 0
       0      .1       0   550.6    .045       0   565.6      .1       0
Bank Sta=550.6,565.6
XS Rating Curve= 0 ,0
Exp/Cntr=0.3,0.1

Type RM Length L Ch R = 1 ,19577.9 ,290,285.3,281.9
XS GIS Cut Line= 3
     1972527.439      383796.517     1972041.157      383578.971
     1971459.599       383360.55
#Sta/Elev= 30
       0 2101.53    98.6 2084.25   138.1 2075.88     217 2056.85     296 2043.27
   394.6 2029.72   525.2 2014.18   532.7 2013.86   540.2 2014.56     582 2024.43
   611.6 2036.41   631.3 2047.07     651    2059   690.5 2086.72   700.4  2092.7
   720.1 2101.32   729.9 2103.89   739.8 2105.17   789.1 2105.12   848.3    2108
   858.1 2109.78     868 2112.95   927.2 2140.38     937 2143.47   956.7 2145.36
  1065.2 2146.87  1084.9 2148.39  1094.8 2150.46  1114.5 2156.97    1154 2173.84
#Mann= 3 , 0 , 0
       0      .1       0   525.2    .045       0   540.2      .1       0
Bank Sta=525.2,540.2
XS Rating Curve= 0 ,0
Exp/Cntr=0.3,0.1

Type RM Length L Ch R = 1 ,19292.6 ,388.6,386.5,384.4
XS GIS Cut Line= 2
      1972595.44      383409.631     1971813.968      383243.624
#Sta/Elev= 30
       0 2093.39      20 2092.36      40 2092.66    49.9 2092.12    59.9  2090.9
    89.9 2085.94   139.8 2076.32   149.8 2073.81   169.8 2067.18   179.8 2062.35
   199.7 2049.42   209.7 2043.48   219.7 2039.44   239.7 2034.94   259.6  2031.9
   279.6 2029.62   459.4 2016.73   479.4 2013.82   519.3 2006.62   530.1  2005.2
   539.3 2005.06   545.1 2005.95   589.2 2013.75   609.2 2017.77   629.1 2023.15
   649.1 2030.01   679.1 2042.44     719 2060.41     739 2070.52   798.9  2102.6
#Mann= 3 , 0 , 0
       0      .1       0   530.1    .045       0   545.1      .1       0
Bank Sta=530.1,545.1
XS Rating Curve= 0 ,0
Exp/Cntr=0.3,0.1

Type RM Length L Ch R = 1 ,18905.8 ,230.8,227.9,227.7
XS GIS Cut Line= 2
     1972579.599      383029.138     1971632.063      382923.253
#Sta/Elev= 30
       0 2087.76    29.8 2083.32   109.2 2072.96   119.2 2071.36     139 2067.35
   178.8 2058.04   248.3 2035.56   268.2 2030.16   278.1 2028.28   337.7 2019.73
   377.4 2015.26   417.1 2009.78   466.8 2000.13   496.6 1993.82   516.4 1990.72
   536.3  1988.8   556.2 1987.65     623 1985.58   635.6 1985.46     638 1985.91
   645.6 1987.34   655.5 1992.75   665.4 1999.45   675.4 2004.04   695.2 2010.72
   734.9 2027.74   754.8 2035.73   824.3 2062.37   913.7 2098.21   953.4 2112.92
#Mann= 3 , 0 , 0
       0      .1       0     623    .045       0     638      .1       0
Bank Sta=623,638
XS Rating Curve= 0 ,0
Exp/Cntr=0.3,0.1

Type RM Length L Ch R = 1 ,18677.9 ,305.1,300,292.4
XS GIS Cut Line= 3
     1972606.529      382774.953     1972073.413      382785.191
     1971457.621      382720.843
#Sta/Elev= 30
       0 2106.15    59.2 2088.07   108.6 2079.42     158 2068.53   266.6 2032.36
   276.5 2029.91   286.4 2028.84   335.7 2028.28   355.5 2026.16   424.6 2010.43
   444.4 2003.84     474 1991.55   513.5 1980.94   525.7 1979.11   533.2 1978.82
   540.7 1979.57   583.2 1988.65   623.1 1994.82     713 1996.23   772.9 2001.34
   812.8 2009.32   842.8 2018.32   862.8  2025.7   952.6 2065.45   982.6 2077.21
  1012.6 2087.19  1062.5 2100.05  1102.4 2112.18  1142.4 2129.11  1152.4 2132.16
#Mann= 3 , 0 , 0
       0     .06       0   525.7    .045       0   540.7     .06       0
Bank Sta=525.7,540.7
XS Rating Curve= 0 ,0
Exp/Cntr=0.3,0.1

Type RM Length L Ch R = 1 ,18377.9 ,301.5,299.9,291.2
XS GIS Cut Line= 3
     1972584.928      382363.195     1972070.039      382491.918
     1971454.575      382637.719
#Sta/Elev= 30
       0 2054.72      30 2051.99    60.1    2047    80.1 2044.36   130.2 2041.14
   180.2 2034.63   260.4 2019.44   380.5 2001.76   460.6 1987.94   480.7 1983.79
   490.7 1980.89   510.7 1973.45   520.7  1971.1   523.2 1971.09   530.7 1971.06
   538.2 1971.77   570.3 1974.93   649.3 1980.66     679 1981.72   718.5 1981.97
   807.4 1984.62   827.2 1987.01   866.8 1995.47   886.5 2000.33   906.3 2006.47
     926 2013.49   955.7 2025.22  1044.6 2062.36  1123.7  2099.6  1163.2 2117.15
#Mann= 3 , 0 , 0
       0     .06       0   523.2    .045       0   538.2     .06       0
Bank Sta=523.2,538.2
XS Rating Curve= 0 ,0
Exp/Cntr=0.3,0.1

Type RM Length L Ch R = 1 ,18077.9 ,256.2,240.4,230.7
XS GIS Cut Line= 3
     1972455.906      382064.036     1971943.819      382228.404
     1971421.182      382561.767
#Sta/Elev= 30
       0 2005.26    39.8 2002.88   139.4 1995.94   189.2 1991.14   358.6 1977.87
   458.1 1972.86   468.1 1971.65   478.1 1969.91   517.9 1961.84   530.3 1960.19
   537.8 1959.91   545.3 1960.39   607.8 1967.42   637.8 1969.48   747.8 1972.43
   777.8 1972.78   787.8 1973.52   797.8 1975.06   827.8  1981.8   857.8 1987.76
   867.8 1990.36   877.8 1993.57   887.8 1997.41   927.8 2014.64  1037.7 2059.43
  1047.7 2063.82  1087.7 2083.38  1117.7 2097.48  1137.7 2106.36  1157.7 2114.26
#Mann= 3 , 0 , 0
       0     .06       0   530.3    .045       0   545.3     .06       0
Bank Sta=530.3,545.3
XS Rating Curve= 0 ,0
Exp/Cntr=0.3,0.1

Type RM Length L Ch R = 1 ,17837.3 ,222.3,224.3,227.7
XS GIS Cut Line= 3
     1972029.301      381674.691     1971752.036        382153.8
     1971384.241      382594.696
#Sta/Elev= 30
       0 2045.67    49.4 2028.79   128.5 2006.43   197.7 1990.03   296.6 1963.59
   306.4 1963.13     346  1964.9   365.7 1963.84   395.4 1961.21   470.2 1951.59
   484.4  1950.4   485.2 1950.43   494.2 1950.73   504.1 1952.26   533.8 1958.36
   553.6 1961.36   573.4 1962.41   622.8 1962.77   642.6 1964.32   692.1 1971.68
   741.6 1982.56   761.4  1987.8   791.1 1997.85   850.5 2024.71   870.3 2033.06
   969.3 2070.03  1028.7    2095  1068.3 2110.78  1107.9 2124.42  1127.7 2128.85
#Mann= 3 , 0 , 0
       0     .06       0   470.2    .045       0   485.2     .06       0
Bank Sta=470.2,485.2
XS Rating Curve= 0 ,0
Exp/Cntr=0.3,0.1

Type RM Length L Ch R = 1 ,17613   ,432.8,435.1,434.4
XS GIS Cut Line= 3
     1971910.363      381575.818     1971577.687      382013.113
     1971228.216      382432.465
#Sta/Elev= 30
       0 2081.49      30 2075.62      50 2069.15    59.9 2064.09    99.9 2038.82
   159.8 2008.82   199.8 1984.37   219.8 1975.28   269.7 1956.42   279.7 1954.52
   289.7 1954.38   349.6 1956.25   369.6 1955.74   489.5 1949.76   535.8 1944.83
   549.4 1943.49   550.8 1943.58   559.4 1944.12   599.1 1954.06   658.6 1960.71
   698.3 1966.16   708.3 1968.34   728.1 1974.28   757.9 1985.21     877    2035
   936.5 2054.69   966.3 2062.85   986.2 2067.07  1045.7  2075.8  1095.3 2084.29
#Mann= 3 , 0 , 0
       0     .06       0   535.8    .045       0   550.8     .06       0
Bank Sta=535.8,550.8
XS Rating Curve= 0 ,0
Exp/Cntr=0.3,0.1

Type RM Length L Ch R = 1 ,17177.9 ,299.3,301,305
XS GIS Cut Line= 3
     1971634.749      381321.711     1971261.554      381719.142
     1970923.254      382161.277
#Sta/Elev= 30
       0 2064.11    39.6 2058.89    59.5 2055.52    79.3 2050.82     109 2042.24
   168.5 2022.28   188.3    2015   267.6 1983.44   297.4 1972.63   317.2 1966.46
     337 1962.44   366.8 1957.62   426.2 1948.63   485.7 1940.74   537.7 1930.92
   545.2 1930.31   552.7 1930.98     575 1935.16     585 1936.04   694.3  1937.9
   714.2  1940.5   783.8 1954.22   833.5 1965.21   883.2 1978.69   942.8 1999.44
   962.7 2005.62   982.6 2010.46  1022.4 2016.68  1042.2 2016.88  1101.9 2013.19
#Mann= 3 , 0 , 0
       0      .1       0   537.7    .045       0   552.7      .1       0
Bank Sta=537.7,552.7
XS Rating Curve= 0 ,0
Exp/Cntr=0.3,0.1

Type RM Length L Ch R = 1 ,16876.9 ,287.3,303.2,319.1
XS GIS Cut Line= 3
     1971467.296      381150.865     1970880.855      381685.382
     1970647.378      381937.355
#Sta/Elev= 30
       0 2012.41    49.6 2008.28    79.4 2005.43   109.1 2002.18   128.9 1999.57
   138.9 1997.66   148.8 1995.37   188.4 1985.19   267.8 1965.66   287.6 1961.11
   396.7 1943.84   446.3 1937.15   476.1 1933.28     486  1932.2   575.3 1924.98
   621.2 1921.63   624.9 1921.45   636.2 1921.72   664.5 1923.31   694.3 1924.54
   753.8 1925.83   803.3 1927.49   881.8 1930.94   930.9 1933.34   940.7 1934.22
   950.5 1935.44   989.8 1941.07  1038.8 1947.19  1087.9 1952.51    1137  1957.1
#Mann= 3 , 0 , 0
       0     .06       0   621.2    .045       0   636.2     .06       0
Bank Sta=621.2,636.2
XS Rating Curve= 0 ,0
Exp/Cntr=0.3,0.1

Type RM Length L Ch R = 1 ,16573.7 ,247.8,241.5,234.3
XS GIS Cut Line= 3
     1971455.292      381136.935     1971129.787      381312.747
     1970322.138       381343.35
#Sta/Elev= 30
       0 2007.84      70 1999.29     110 1993.26     120 1991.44     180 1978.76
     250 1960.93     260 1958.64     360 1941.82   409.9 1934.07   459.8 1925.02
   469.7 1923.81   479.7 1923.29   509.6 1922.73   529.6 1921.97   609.4 1916.53
   638.5 1914.22   649.3 1913.64   653.5 1913.64     799 1918.31   828.9 1919.66
   848.9 1921.24   908.8 1927.94   918.8 1929.24   938.7 1932.52   958.7 1937.03
   988.6 1945.21  1058.4 1966.98  1078.4 1973.88  1118.3 1988.97  1178.2 2010.71
#Mann= 3 , 0 , 0
       0     .06       0   638.5    .045       0   653.5     .06       0
Bank Sta=638.5,653.5
XS Rating Curve= 0 ,0
Exp/Cntr=0.3,0.1

Type RM Length L Ch R = 1 ,16332.5 ,262.5,265.9,272.2
XS GIS Cut Line= 3
     1971401.627      381062.288     1971076.335       381056.18
      1970302.05      381234.861
#Sta/Elev= 30
       0 1993.82      69 1980.48   177.5 1956.28     207 1950.98     276 1937.58
   305.6 1932.74   325.4 1930.03   355.2 1927.37   365.1 1925.45   394.9 1918.51
   404.8 1916.81   454.5 1911.94   474.3  1909.5   491.3  1908.6   494.2 1908.54
   506.3 1908.74   553.8 1909.43   603.5 1912.58   643.2 1913.76   663.1  1913.6
   692.9 1912.62   722.7 1912.62   742.5 1914.04   762.4 1916.11   802.1 1921.29
   871.7 1935.83   891.5 1941.55   941.2 1958.25   990.9 1975.54    1120 2024.67
#Mann= 3 , 0 , 0
       0     .06       0   491.3    .045       0   506.3     .06       0
Bank Sta=491.3,506.3
XS Rating Curve= 0 ,0
Exp/Cntr=0.3,0.1

Type RM Length L Ch R = 1 ,16065.6 ,421.6,414,406
XS GIS Cut Line= 3
     1971355.529      380809.229     1970879.328      380918.733
     1970213.474      380961.494
#Sta/Elev= 30
       0 1964.12    49.9 1958.35   139.6  1947.2   219.4 1935.78   259.3 1930.84
     349 1922.93   418.8 1915.64   468.7 1911.98   558.3 1901.83   588.2 1898.84
   605.7 1897.98   608.1 1897.94   618.1 1898.94   620.7 1899.56   657.9 1909.89
   667.9 1912.28   677.8 1913.99   707.7 1916.83   717.7 1918.31   737.6 1922.71
   757.5 1927.79   797.4 1939.19   837.2 1952.47     887 1967.88   946.7 1987.57
   956.7 1991.59  1026.4 2023.77  1106.1 2063.14  1135.9 2076.66  1155.9 2085.05
#Mann= 3 , 0 , 0
       0      .1       0   605.7    .045       0   620.7      .1       0
Bank Sta=605.7,620.7
XS Rating Curve= 0 ,0
Exp/Cntr=0.3,0.1

Type RM Length L Ch R = 1 ,15651.2 ,275.8,259.7,243.7
XS GIS Cut Line= 2
     1971088.553      380430.032     1970187.015      380838.425
#Sta/Elev= 30
       0 1967.88      20  1963.4      50 1955.08      70 1950.49   199.9 1926.03
   269.9 1911.56   279.9 1908.42   289.9 1900.97   299.9 1892.54   305.3 1891.01
   309.9 1889.71   320.3 1890.51   349.9 1894.49   469.9 1902.21   489.9 1903.12
   529.8 1902.81   539.8 1903.46   549.8 1905.04   559.8 1907.79   589.8 1919.22
   599.8 1922.38   629.8  1930.8   659.8 1938.18   679.8 1944.92   729.8 1968.18
   789.8 1999.46   829.8 2018.38   889.8 2041.17   939.7 2058.47   989.7 2078.11
#Mann= 3 , 0 , 0
       0      .1       0   305.3    .045       0   320.3      .1       0
Bank Sta=305.3,320.3
XS Rating Curve= 0 ,0
Exp/Cntr=0.3,0.1

Type RM Length L Ch R = 1 ,15391.4 ,303.4,314.6,330.7
XS GIS Cut Line= 3
     1970822.822      379938.277     1970520.439       380588.86
     1970265.398      380726.307
#Sta/Elev= 30
       0 1970.74   159.4 1938.92   229.2 1927.08   298.9 1917.93   338.8 1913.49
   378.6 1907.28   398.6 1906.32   468.3 1904.35   478.3 1902.43   488.2  1897.5
   498.2 1891.18   508.2 1886.88   509.7 1886.69   518.1 1885.62   524.7 1886.04
     558 1890.21   617.8 1900.29   677.6 1908.93   777.4  1928.2   797.3 1932.68
   807.3 1935.45   827.3 1942.18   847.3  1950.9   857.3 1955.96   877.3 1967.28
   917.2 1992.28   937.2 2004.08   947.2 2009.33   967.2 2018.64  1007.1 2035.19
#Mann= 3 , 0 , 0
       0      .1       0   509.7    .045       0   524.7      .1       0
Bank Sta=509.7,524.7
XS Rating Curve= 0 ,0
Exp/Cntr=0.3,0.1

Type RM Length L Ch R = 1 ,15076.8 ,291.7,299.8,304.1
XS GIS Cut Line= 3
     1970832.591      379878.145     1970360.301      380227.279
     1969868.024      380446.069
#Sta/Elev= 30
       0 1979.89    39.8  1971.7   139.4 1946.42   189.1 1934.66     229 1926.12
   318.6 1908.48   378.3 1899.52   418.1 1895.72   457.9 1894.36   507.7 1895.19
   517.6 1892.53   537.6  1881.4   547.5 1877.98   579.8 1873.39   587.3 1872.59
   594.8 1872.68   597.3 1872.71   607.3 1875.04   627.2 1883.86   667.1 1899.08
     707 1912.56     727 1918.72   816.8  1938.9   836.7 1944.17   926.5 1970.16
   946.5  1975.1   966.4 1979.03   986.4  1984.2  1046.2 2001.66    1126 2027.66
#Mann= 3 , 0 , 0
       0      .1       0   579.8    .045       0   594.8      .1       0
Bank Sta=579.8,594.8
XS Rating Curve= 0 ,0
Exp/Cntr=0.3,0.1

Type RM Length L Ch R = 1 ,14776.8 ,305.9,293.2,279.3
XS GIS Cut Line= 3
     1970796.895      379800.927     1970247.012      379959.427
     1969717.766       380082.83
#Sta/Elev= 30
       0 1983.42    39.5 1974.66    78.9 1965.08   226.9 1925.51   266.4 1915.88
   404.5 1892.32   434.1 1889.99   522.9 1885.85   532.8  1884.4   542.7 1880.72
   562.4 1869.75   564.8 1869.06   572.3 1866.91   579.8  1866.8   582.2 1866.77
     592 1868.54   641.4 1882.64   651.3 1884.95   750.1 1898.06   769.9 1903.21
   829.2  1921.8   937.9 1957.31   947.7 1961.32   957.6 1966.33   977.4 1977.52
  1016.9 1997.74  1056.4 2016.49    1096 2033.24  1105.8 2036.05  1115.7 2037.01
#Mann= 3 , 0 , 0
       0      .1       0   564.8    .045       0   579.8      .1       0
Bank Sta=564.8,579.8
XS Rating Curve= 0 ,0
Exp/Cntr=0.3,0.1

Type RM Length L Ch R = 1 ,14483.6 ,301.7,306.8,311.8
XS GIS Cut Line= 3
     1970531.609      379289.606     1970024.102      379863.445
     1969683.273      379992.601
#Sta/Elev= 30
       0 2026.18    29.8 2023.14    39.8 2021.25    49.7 2015.87    79.6 1993.78
    89.5 1987.44    99.5 1982.29     189 1954.62   208.9 1946.93   238.8 1932.12
   248.7 1928.93   278.6 1925.79     398 1901.73   417.8 1896.63   487.5 1873.64
   535.5 1861.33   537.2    1861   550.5 1862.02     587 1868.08   656.6  1876.6
   736.2 1881.82   766.1 1884.77   805.5 1891.76   844.9 1901.94   884.3 1915.52
   992.6 1958.87  1022.2 1974.61  1110.8 2024.68  1120.7  2029.5  1130.5 2032.35
#Mann= 3 , 0 , 0
       0      .1       0   535.5    .045       0   550.5      .1       0
Bank Sta=535.5,550.5
XS Rating Curve= 0 ,0
Exp/Cntr=0.3,0.1

Type RM Length L Ch R = 1 ,14176.8 ,297.2,299.9,299.8
XS GIS Cut Line= 3
     1970430.661      379140.258     1969988.086      379457.403
     1969538.889      379780.823
#Sta/Elev= 30
       0 1992.01    19.8 1982.29    29.7 1978.72    39.6 1976.06   148.5 1950.61
   227.7 1926.23   267.3 1919.09     297 1910.82   336.6  1901.2   376.2 1889.25
   455.4 1868.49   465.3 1866.24     495 1864.08   504.9 1861.78   514.8 1858.55
     537 1849.42   544.5 1847.63     552 1847.61   564.2 1849.33   613.7 1861.25
   633.4 1864.85   761.9 1873.56   781.7 1875.63   791.6 1877.78   801.5  1881.1
   870.6 1908.88   969.5 1947.45   979.4 1951.83  1028.8 1976.72    1098  2008.2
#Mann= 3 , 0 , 0
       0      .1       0     537    .045       0     552      .1       0
Bank Sta=537,552
XS Rating Curve= 0 ,0
Exp/Cntr=0.3,0.1

Type RM Length L Ch R = 1 ,13876.8 ,306.2,300,291.9
XS GIS Cut Line= 3
     1970286.875      378961.859     1969810.902      379223.645
     1969358.075      379556.138
#Sta/Elev= 30
       0  1965.4    69.1 1948.51    88.9 1941.88   148.2 1919.99   167.9 1914.48
   266.7 1895.41   325.9 1882.59   365.4 1873.04   385.2 1870.11   424.7 1868.41
   434.6 1866.68   444.4 1862.93   464.2 1853.18   474.1 1850.92   503.7 1846.45
   535.7 1840.49   543.2 1839.55   550.7 1839.67   562.9 1841.55   582.6 1847.29
   602.4 1852.03   612.2 1853.24   681.2 1856.81   720.6 1859.96     760 1865.78
   809.3 1876.49   888.2  1902.7   947.3 1923.22  1055.7 1962.64    1105 1982.38
#Mann= 3 , 0 , 0
       0      .1       0   535.7    .045       0   550.7      .1       0
Bank Sta=535.7,550.7
XS Rating Curve= 0 ,0
Exp/Cntr=0.3,0.1

Type RM Length L Ch R = 1 ,13576.8 ,267.8,282.2,301.5
XS GIS Cut Line= 3
     1969993.076      378618.591     1969596.899      379033.116
     1969298.063       379494.33
#Sta/Elev= 30
       0  1940.4    49.4 1924.94    69.2 1922.18   108.8 1919.63   118.6 1917.16
   138.4 1907.58   158.2 1901.45     178 1896.27   286.7 1871.36   355.9 1857.28
   395.4 1850.73   444.9 1846.84   484.4 1842.21   565.9 1830.16   573.4 1829.73
   580.9 1830.41   593.4 1832.89   623.4 1840.34   643.3  1844.2   743.3 1855.08
   763.2 1858.37   773.2 1860.86   783.2 1864.22   813.2 1876.88   833.2 1880.74
   843.2 1883.61   943.1  1919.4    1013  1943.2    1083 1964.23    1123 1977.91
#Mann= 3 , 0 , 0
       0      .1       0   565.9    .045       0   580.9      .1       0
Bank Sta=565.9,580.9
XS Rating Curve= 0 ,0
Exp/Cntr=0.3,0.1

Type RM Length L Ch R = 1 ,13294.6 ,162.1,159.3,156.5
XS GIS Cut Line= 3
     1969940.631      378557.509     1969665.213      378818.847
     1968867.353      378925.977
#Sta/Elev= 30
       0  1950.5      40 1939.56    79.9 1924.92    89.9 1922.33   129.9 1919.91
   139.9 1918.64   149.9 1916.05   259.8 1876.88   279.8 1870.73   379.7 1851.52
   399.6 1846.29   419.4 1839.71   439.3 1836.93   469.1 1835.01   518.8 1834.07
   558.6 1825.13   608.3 1821.77   618.2 1821.24   628.1 1821.26   638.1 1822.36
   667.9  1828.6   727.5 1833.44     817 1843.57   846.8 1848.27   876.6 1855.73
     976 1886.98  1075.4 1935.58  1144.9 1972.44  1164.8 1981.75  1184.7 1988.85
#Mann= 3 , 0 , 0
       0      .1       0   608.3    .045       0   628.1      .1       0
Bank Sta=608.3,628.1
XS Rating Curve= 0 ,0
Exp/Cntr=0.3,0.1

Type RM Length L Ch R = 1 ,13135.1 ,166.2,158.3,152.5
XS GIS Cut Line= 2
     1969666.231      378634.397     1969058.409      378793.225
#Sta/Elev= 30
       0 1871.33    19.9 1866.64   119.7 1844.08   129.6 1842.28   139.6 1841.24
   159.6  1840.1   169.5 1839.26   179.5 1837.74   189.5 1835.45   209.4    1830
   219.4 1826.63   229.4 1821.85   239.3 1817.89   247.2 1817.01   249.3 1816.78
   262.2 1818.06   299.2  1823.5   309.1 1824.77   319.1 1825.64   329.1 1826.01
     369  1826.1   468.7  1828.1   488.6  1829.3   498.6 1830.24   508.6 1831.54
   518.5 1833.43   538.5 1838.22   548.4 1840.92   558.4 1844.19   628.2 1868.64
#Mann= 3 , 0 , 0
       0      .1       0   247.2    .045       0   262.2      .1       0
Bank Sta=247.2,262.2
XS Rating Curve= 0 ,0
Exp/Cntr=0.3,0.1

Type RM Length L Ch R = 1 ,12976.8 ,268.8,261.6,253.2
XS GIS Cut Line= 3
     1969776.054      378263.606     1969329.763       378570.62
     1968832.396      378849.889
#Sta/Elev= 30
       0 1905.42    59.1 1896.28   108.3 1887.58   137.9  1885.7   147.7 1882.97
   177.3 1871.38     197 1866.61   285.6 1852.25     453  1829.8   472.8 1825.14
   534.2 1807.79   541.7 1806.33   549.2 1806.69   551.7 1806.81   581.7 1815.83
   601.7 1819.35   641.8 1824.85   721.8 1827.47   781.9 1832.69   801.9 1835.84
   821.9 1840.08   851.9 1848.14     922 1872.14     962 1884.28     972 1889.19
    1042 1928.71  1062.1 1941.57  1092.1 1962.26  1102.1 1968.69  1112.1 1974.11
#Mann= 3 , 0 , 0
       0      .1       0   534.2    .045       0   549.2      .1       0
Bank Sta=534.2,549.2
XS Rating Curve= 0 ,0
Exp/Cntr=0.3,0.1

Type RM Length L Ch R = 1 ,12715.2 ,332.8,336.7,338.8
XS GIS Cut Line= 3
     1969478.697      377946.825     1969151.183      378383.513
     1968804.938      378806.724
#Sta/Elev= 30
       0 1869.51    29.8 1861.19    49.6 1857.22    79.4 1854.04     129 1851.54
   178.6 1845.34   198.5 1841.52   238.2 1832.08     258 1829.02   357.3  1819.1
   426.8 1815.34   436.7  1813.2   456.5 1805.65   466.5 1803.65   496.2 1803.84
   506.2 1802.49   541.3 1791.85   545.9 1790.87   556.3 1791.38   565.7 1793.66
   625.4 1812.13     685 1820.33   734.8 1829.58   794.4 1835.01     864 1854.49
   943.5 1879.14   993.2 1897.87  1062.8 1928.45  1072.8 1933.92  1092.7 1947.16
#Mann= 3 , 0 , 0
       0      .1       0   541.3    .045       0   556.3      .1       0
Bank Sta=541.3,556.3
XS Rating Curve= 0 ,0
Exp/Cntr=0.3,0.1

Type RM Length L Ch R = 1 ,12378.3 ,205.6,200.8,196.9
XS GIS Cut Line= 3
      1969312.92      377814.981     1968896.992      378166.165
     1968505.721      378560.345
#Sta/Elev= 30
       0 1908.91    29.7    1900   257.3 1840.68   277.1    1837   306.8 1833.99
   316.7 1831.57   336.5 1824.18   366.2 1810.58     386 1803.48   405.8 1799.94
   504.8 1793.49   514.7  1791.1   534.5 1781.56   544.4 1777.76   548.6 1777.34
   554.3 1776.77   563.6    1779     594 1793.87   613.8 1802.23   693.1 1824.24
   742.7 1835.59   772.5 1845.92   802.2 1860.09   841.9 1885.23   861.7 1895.69
   970.8  1937.4  1060.1 1978.62    1070 1979.86  1079.9 1978.82  1099.8 1974.77
#Mann= 3 , 0 , 0
       0      .1       0   548.6    .045       0   563.6      .1       0
Bank Sta=548.6,563.6
XS Rating Curve= 0 ,0
Exp/Cntr=0.3,0.1

Type RM Length L Ch R = 1 ,12178   ,427.4,422.7,418.8
XS GIS Cut Line= 2
     1969098.072      377560.988     1968432.948      378475.114
#Sta/Elev= 30
       0  1981.4     110  1918.4   140.1 1902.43   150.1 1898.38   210.1  1879.1
   300.1 1853.43   370.2 1831.29   400.2 1825.86   410.2 1822.92   430.2 1813.95
   460.2 1797.01   480.2 1788.24   490.2 1785.88   520.2 1782.36   550.2 1769.06
   554.6 1768.18   560.2 1767.06   569.6 1767.76   600.3 1775.94   630.3 1778.54
   640.3 1780.96   840.4 1846.22   860.4 1854.76   920.4 1886.81  1050.5 1949.58
  1080.5 1968.14  1090.5 1972.84  1100.5 1975.06  1110.5  1975.1  1130.5 1971.87
#Mann= 3 , 0 , 0
       0      .1       0   554.6    .045       0   569.6      .1       0
Bank Sta=554.6,569.6
XS Rating Curve= 0 ,0
Exp/Cntr=0.3,0.1

Type RM Length L Ch R = 1 ,11754.3 ,270.3,277.6,286.3
XS GIS Cut Line= 3
     1968652.462      377342.899      1968415.14      377936.037
     1968196.686      378418.176
#Sta/Elev= 30
       0  1920.6    39.9 1899.68    59.9 1892.08   179.7 1857.61   299.5 1824.57
   429.2 1784.03   439.2 1782.23   499.1  1779.5   519.1 1776.61     539 1771.51
   588.9 1755.06   618.9 1747.78   638.3 1741.56   648.8 1739.42   653.3 1739.41
   658.8 1739.39   668.8 1740.92   688.8 1750.61   728.7 1778.34   768.7    1802
   868.6 1865.37   958.4 1917.72  1018.4 1951.02  1028.4 1953.96  1038.3  1954.7
  1078.3 1953.84  1088.3 1955.13  1098.3 1959.07  1138.2 1980.49  1168.2  1991.5
#Mann= 3 , 0 , 0
       0      .1       0   638.3    .045       0   653.3      .1       0
Bank Sta=638.3,653.3
XS Rating Curve= 0 ,0
Exp/Cntr=0.3,0.1

Type RM Length L Ch R = 1 ,11476.6 ,299.5,300,295.8
XS GIS Cut Line= 3
     1968607.539      377306.032     1968250.111       377718.98
     1967848.066      378104.551
#Sta/Elev= 30
       0 1927.92    39.7 1903.72    59.6 1893.07     139 1864.43   258.2 1824.76
   397.2 1785.41   417.1 1778.41   446.8 1766.68   456.8 1763.74   486.6  1758.6
   516.4 1748.08   536.2 1739.03   546.2 1735.47   556.1  1734.6     566 1736.38
   585.9 1744.07   635.7 1758.56   715.3 1784.96   745.1 1795.69   774.9 1807.53
   814.7  1827.2   874.4  1859.1     954 1896.75  1003.7 1922.02  1013.7 1926.08
  1023.6 1927.04  1063.4 1926.28  1073.4 1927.85  1083.3 1932.34  1103.2 1945.23
#Mann= 3 , 0 , 0
       0      .1       0   546.2    .045       0     566      .1       0
Bank Sta=546.2,566
XS Rating Curve= 0 ,0
Exp/Cntr=0.3,0.1

Type RM Length L Ch R = 1 ,11176.6 ,329.8,328.6,331
XS GIS Cut Line= 3
     1968375.881      377137.615     1968009.709      377541.666
     1967689.314      377988.746
#Sta/Elev= 30
       0 1945.77    29.7 1929.25    69.4 1908.74     119 1885.53   188.4 1851.18
   247.9 1822.96   267.7 1815.82   366.8 1784.87   396.6 1776.94   426.3 1770.52
   446.2 1762.33   495.7 1737.56   505.6 1733.89   537.8 1724.69   545.3 1723.02
   552.8 1722.81   555.3 1722.74   565.3 1724.52   585.3 1732.08   605.3  1737.9
   695.3 1754.19   705.3 1756.55   715.3 1760.28   855.3 1830.82   995.3 1911.42
  1005.3 1916.43  1015.3 1918.95  1055.3 1918.41  1065.3 1920.46  1095.3 1935.83
#Mann= 3 , 0 , 0
       0      .1       0   537.8    .045       0   552.8      .1       0
Bank Sta=537.8,552.8
XS Rating Curve= 0 ,0
Exp/Cntr=0.3,0.1

Type RM Length L Ch R = 1 ,10848   ,270.3,271.4,271.6
XS GIS Cut Line= 3
     1968081.654      376927.161     1967742.175      377356.252
     1967379.017      377763.698
#Sta/Elev= 30
       0 1912.46    39.8 1895.75    69.6 1882.31   139.3 1856.38   218.9 1828.96
   288.5 1807.46   308.4 1800.55   417.8 1757.64   487.4 1724.14   497.4 1721.14
   527.2 1714.91   544.2 1710.15   557.1 1708.13   559.2 1708.23     567 1708.59
   586.8 1713.48   656.3 1735.46   676.2 1743.02   775.4 1790.83   914.3 1851.19
   924.2 1856.17   944.1 1868.35   993.7 1903.59  1003.6  1907.5  1013.6 1908.26
  1043.3 1906.29  1063.2 1906.13  1073.1 1907.46    1083 1910.19  1092.9 1913.88
#Mann= 3 , 0 , 0
       0      .1       0   544.2    .045       0   559.2      .1       0
Bank Sta=544.2,559.2
XS Rating Curve= 0 ,0
Exp/Cntr=0.3,0.1

Type RM Length L Ch R = 1 ,10576.6 ,303.8,300,294.4
XS GIS Cut Line= 3
     1967898.421      376777.804     1967533.653      377184.104
     1967166.017      377587.782
#Sta/Elev= 30
       0 1951.44    49.6  1919.5    89.4 1895.43   109.2 1884.58   148.9 1864.65
   198.6 1835.93   228.3 1820.94   258.1 1808.77   317.7 1789.39     417 1753.55
   436.8 1744.08   466.6 1727.12   486.4 1716.93   496.4 1712.98   538.5 1699.41
     546 1698.08   553.5  1698.2   565.9 1700.96   585.7 1710.91   625.4 1727.14
   645.3  1734.4   794.2 1776.77     814 1783.59   923.2 1829.04  1012.6 1881.35
  1022.5 1886.86  1032.4 1891.33  1042.4 1893.67  1052.3 1893.79    1092 1891.62
#Mann= 3 , 0 , 0
       0      .1       0   538.5    .045       0   553.5      .1       0
Bank Sta=538.5,553.5
XS Rating Curve= 0 ,0
Exp/Cntr=0.3,0.1

Type RM Length L Ch R = 1 ,10276.6 ,303.7,300,294.4
XS GIS Cut Line= 3
     1967582.339      376547.295     1967290.966      377008.638
     1967033.211      377492.205
#Sta/Elev= 30
       0 1924.78    99.2 1874.52     119  1865.7   148.8 1854.37   158.7 1849.69
   208.3 1821.74   228.2 1811.88     248 1803.65   267.9  1796.5   307.6 1786.15
   327.4 1780.27   436.5 1740.93   515.9 1703.12   535.7  1689.8   545.6 1685.22
   555.6 1684.56   565.6 1686.74   585.5 1694.12   625.4 1706.65     725 1733.28
   774.8 1748.75   824.6 1765.37   894.4 1793.86   944.2  1815.6   974.1 1832.82
  1043.8 1875.79  1053.8 1881.42  1063.7 1884.79  1073.7 1885.07  1093.6  1883.5
#Mann= 3 , 0 , 0
       0      .1       0   545.6    .045       0   555.6      .1       0
Bank Sta=545.6,555.6
XS Rating Curve= 0 ,0
Exp/Cntr=0.3,0.1

Type RM Length L Ch R = 1 ,9976.6  ,294.9,303.5,317.8
XS GIS Cut Line= 3
     1967221.857      376405.402     1967006.705       376917.24
     1966877.712       377446.11
#Sta/Elev= 30
       0 1779.46    79.3 1769.56   287.5 1752.82     347 1744.17   366.8 1739.91
   376.8 1736.36   396.6 1727.26   436.2 1706.11   446.2 1701.74   456.1 1698.74
   495.7 1690.13   535.4 1677.43   547.7 1675.16   555.2 1674.88   562.7 1675.79
   614.6 1685.79     674 1703.72   713.6 1719.31   832.4 1769.94   891.7 1793.77
   931.3 1812.36   970.9 1834.05   990.7 1846.82  1000.6 1854.22  1020.4 1871.48
  1030.3 1877.31  1040.2 1879.28  1079.8 1876.45  1089.7 1877.91  1099.6 1882.92
#Mann= 3 , 0 , 0
       0      .1       0   547.7    .045       0   562.7      .1       0
Bank Sta=547.7,562.7
XS Rating Curve= 0 ,0
Exp/Cntr=0.3,0.1

Type RM Length L Ch R = 1 ,9673.2  ,293.3,301,306.6
XS GIS Cut Line= 3
      1967146.77      376362.575     1966742.326      376786.455
      1966327.76      377130.862
#Sta/Elev= 30
       0    1760    49.6 1750.42   158.9 1733.22     278 1712.61   307.8 1708.83
   466.7 1694.74   546.2 1677.92   581.7 1667.65   595.9 1665.96   596.7 1666.14
   605.8 1668.18   655.7 1694.32   675.7 1709.29   715.6 1741.57   735.6 1755.73
   765.5 1772.26   805.4 1788.19   815.4 1793.28   915.2 1857.33   925.2 1861.52
   935.2 1862.17   955.2 1859.08   975.1 1858.14   995.1 1858.62  1005.1  1861.8
    1015 1868.42    1045 1893.48    1055 1900.75  1074.9 1911.66  1124.8 1935.25
#Mann= 3 , 0 , 0
       0      .1       0   581.7    .045       0   596.7      .1       0
Bank Sta=581.7,596.7
XS Rating Curve= 0 ,0
Exp/Cntr=0.3,0.1

Type RM Length L Ch R = 1 ,9372    ,346,330.8,315.6
XS GIS Cut Line= 3
     1967095.998      376290.688     1966431.644      376607.477
     1966168.409      376900.653
#Sta/Elev= 30
       0 1749.86    39.8 1741.25   258.6 1711.18   437.6 1697.39   447.6 1695.63
   457.5 1692.48   477.4  1683.5   497.3 1673.25   517.2 1661.15   527.2 1656.49
   537.1 1655.03   538.3 1655.07   553.3 1655.71   586.8 1658.76   646.5 1671.53
     736 1687.12   814.8 1706.42   824.7 1710.47   834.5  1715.9   883.8 1746.63
   942.9 1784.53    1002 1825.74  1021.7 1837.39  1031.5 1841.65  1051.2 1846.63
  1070.9 1848.33  1100.5 1846.85  1110.3 1848.93  1120.2  1854.7    1130 1863.57
#Mann= 3 , 0 , 0
       0      .1       0   538.3    .045       0   553.3      .1       0
Bank Sta=538.3,553.3
XS Rating Curve= 0 ,0
Exp/Cntr=0.3,0.1

Type RM Length L Ch R = 1 ,9041.1  ,272.6,271.5,269.2
XS GIS Cut Line= 3
     1966526.497       375845.19     1966411.281      376228.056
     1966102.202      376852.421
#Sta/Elev= 30
       0 1874.62      50 1864.83      70 1859.61      80 1855.21   159.9 1811.66
   239.9 1769.65   329.9 1724.86   409.8 1689.18   479.4 1660.78   529.2 1642.13
   539.2 1639.78   543.3  1639.6   549.1 1639.34   558.3  1640.2   588.9  1644.7
   598.9 1647.37   618.8 1656.02   628.7  1659.2   718.3 1674.27   738.2 1678.94
   748.2 1682.56   807.9 1708.06   857.6 1734.84   947.2 1780.95  1046.7 1828.08
  1056.7 1832.29  1066.6 1835.08  1076.6 1836.49  1086.6 1838.81  1096.5 1844.45
#Mann= 3 , 0 , 0
       0      .1       0   543.3    .045       0   558.3      .1       0
Bank Sta=543.3,558.3
XS Rating Curve= 0 ,0
Exp/Cntr=0.3,0.1

Type RM Length L Ch R = 1 ,8769.5  ,311.8,300.1,291.4
XS GIS Cut Line= 3
     1966310.412      375765.797     1966091.662      376265.602
     1965899.913      376778.767
#Sta/Elev= 30
       0 1859.05    19.8 1861.31    29.8 1860.77    49.6 1856.47    69.4 1850.53
    79.4 1844.36    89.3 1835.42    99.2 1828.19   109.1 1822.77   158.7  1797.7
   198.4 1779.75   347.2 1702.58     377 1689.35   416.6 1673.69   446.4  1663.4
   486.1 1651.92   538.1  1631.1   553.1 1629.41   555.5 1629.37   645.2 1636.52
   655.1  1639.1   704.9 1656.92   744.8 1664.37   754.8 1667.52   854.4 1714.55
     934 1756.86  1053.6 1816.74  1073.5 1825.99  1083.4  1827.3  1093.4 1825.28
#Mann= 3 , 0 , 0
       0      .1       0   538.1    .045       0   553.1      .1       0
Bank Sta=538.1,553.1
XS Rating Curve= 0 ,0
Exp/Cntr=0.3,0.1

Type RM Length L Ch R = 1 ,8469.5  ,302.2,300,294.1
XS GIS Cut Line= 3
     1965741.879      375673.135     1965802.123      376215.339
     1965813.178      376763.833
#Sta/Elev= 30
       0 1912.42    19.8 1895.96    69.4 1847.39    79.4 1839.24    89.3 1836.03
     119 1836.92     129 1835.69   178.5 1824.64   188.5 1820.54   208.3 1804.21
   218.2 1797.25   317.4 1735.33   436.4 1665.74   476.1 1639.76   505.9 1623.66
   515.8 1619.55   525.7 1617.29     538 1616.61   545.5 1616.53     553 1616.73
   645.3 1624.41   665.2 1627.42   705.1 1640.63   735.1 1652.84     765 1659.47
     775 1662.89   854.8 1706.55   914.6  1729.3   974.4 1753.98  1094.2 1815.32
#Mann= 3 , 0 , 0
       0      .1       0     538    .045       0     553      .1       0
Bank Sta=538,553
XS Rating Curve= 0 ,0
Exp/Cntr=0.3,0.1

Type RM Length L Ch R = 1 ,8169.5  ,261.8,263.8,267.6
XS GIS Cut Line= 3
     1965391.602      375721.649     1965505.119      376255.178
     1965660.178      376781.817
#Sta/Elev= 30
       0 1914.02    49.6 1886.61    59.5 1879.41    79.3 1859.44     119 1815.19
   128.9 1809.21   138.8 1808.78   178.5 1815.29   188.4 1814.96     238 1799.87
   257.9 1787.06   297.5 1755.05   376.9 1695.76   436.4 1654.65   495.9 1620.63
     538 1610.03     553 1608.38   555.4 1608.25   645.3 1616.26   665.2 1621.91
   735.1 1649.38   765.1 1655.93     775 1659.72     785 1666.34     825 1697.96
   854.9 1715.35   934.8 1749.31  1004.6 1782.47  1064.5 1806.25  1094.5 1813.78
#Mann= 3 , 0 , 0
       0      .1       0     538    .045       0     553      .1       0
Bank Sta=538,553
XS Rating Curve= 0 ,0
Exp/Cntr=0.3,0.1

Type RM Length L Ch R = 1 ,7905.7  ,374.1,359.7,345.3
XS GIS Cut Line= 3
     1965207.856      375860.173     1965293.379      376566.752
     1965465.927      376864.745
#Sta/Elev= 30
       0 1853.99     9.9 1843.13    39.5 1806.67    49.4 1796.86    59.3 1792.94
    98.8 1794.98   138.4 1791.17   158.2 1788.17     168 1783.56   187.8  1767.9
   306.4 1663.63   355.9 1626.42   375.6 1614.15   385.5 1611.43   395.4 1610.42
   504.6 1601.91   519.6 1600.52   523.9 1600.27   533.8 1600.82   642.5 1621.36
   662.3 1628.34     692 1641.97   721.6 1650.05   731.4  1653.8   741.2 1659.29
   800.3 1697.86   839.6 1720.56   947.9 1762.29  1046.2 1805.28  1056.1 1808.46
#Mann= 3 , 0 , 0
       0      .1       0   504.6    .045       0   519.6      .1       0
Bank Sta=504.6,519.6
XS Rating Curve= 0 ,0
Exp/Cntr=0.3,0.1

Type RM Length L Ch R = 1 ,7546    ,116.8,109,101.1
XS GIS Cut Line= 3
     1965025.804      375770.286     1964908.527       376302.04
     1965413.518      376817.211
#Sta/Elev= 30
       0 1832.75    19.8 1818.34    39.6 1800.54    49.5 1793.68    59.4 1789.82
    79.2  1787.8   158.4 1785.93   287.1 1786.13   316.8 1781.35   356.4 1769.48
   376.2  1760.3   405.9 1743.31   445.5 1724.59   485.1 1695.16   544.5 1656.87
   574.2 1634.83   623.6 1601.21   643.4 1592.28   656.7 1589.78   671.7 1588.73
     673 1588.69   712.5 1594.84   791.6 1599.46   929.9 1616.46   939.8 1620.45
   969.5 1637.81  1018.9 1652.19  1078.2 1686.39  1137.5 1722.83  1265.9  1776.6
#Mann= 3 , 0 , 0
       0      .1       0   656.7    .045       0   671.7      .1       0
Bank Sta=656.7,671.7
XS Rating Curve= 0 ,0
Exp/Cntr=0.3,0.1

Type RM Length L Ch R = 1 ,7437    ,255.7,267.9,280.1
XS GIS Cut Line= 4
     1964913.045      376058.061      1964877.92      376452.075
     1965047.743      376536.987     1965343.713      376826.237
#Sta/Elev= 30
       0  1780.4    98.9 1758.22   118.7 1752.29   138.4 1742.91   158.2 1731.13
   207.7 1692.79   237.4  1671.6   247.2 1665.55   316.5 1631.84   385.7 1602.12
   395.6 1599.04   435.6 1593.66   465.1 1586.95   475.5 1585.75   480.1 1586.12
   525.5 1593.25   585.4 1599.08     684 1611.16   703.7 1615.02   713.5 1620.06
   733.2    1633   743.1 1638.07     753  1641.4   792.4 1649.39   812.1 1660.76
   851.5  1687.6   871.2 1699.75   890.9  1708.9   940.2 1728.34   999.3 1754.02
#Mann= 3 , 0 , 0
       0      .1       0   465.1    .045       0   480.1      .1       0
Bank Sta=465.1,480.1
XS Rating Curve= 0 ,0
Exp/Cntr=0.3,0.1

Type RM Length L Ch R = 1 ,7169.1  ,187.3,216.9,246.4
XS GIS Cut Line= 5
     1964882.501      376059.588     1964830.744      376549.575
     1964851.894      376714.932     1964951.289      376867.439
     1965256.726      377124.007
#Sta/Elev= 30
       0 1770.55    88.7 1750.14   108.4 1746.64     138 1743.59   147.8 1740.64
   167.5  1729.6   236.5 1683.95   256.2 1671.98     335 1630.05   394.2 1600.91
   413.9 1597.08   531.9  1586.1   551.6  1585.1     630  1584.6   649.6 1581.74
   677.7 1575.66   688.2 1574.82   692.7  1575.5   697.7 1576.26   726.5 1587.07
   774.4 1601.03   812.7 1614.43   881.3 1625.89   931.2 1636.93   961.1  1644.3
  1060.8 1673.63  1090.8 1684.44  1180.5 1720.08  1210.4 1733.89  1240.4 1750.39
#Mann= 3 , 0 , 0
       0      .1       0   677.7    .045       0   692.7      .1       0
Bank Sta=677.7,692.7
XS Rating Curve= 0 ,0
Exp/Cntr=0.3,0.1

Type RM Length L Ch R = 1 ,6952.2  ,287.5,293.9,300.2
XS GIS Cut Line= 3
     1964847.376      376203.144     1964768.026      376617.659
     1964359.911      377080.241
#Sta/Elev= 30
       0 1733.67    19.6 1728.29    39.3 1718.77     108  1677.5   176.7 1640.06
   215.9 1613.73   225.7 1608.65   235.6 1605.05   245.4 1602.43     265 1599.35
   333.7 1592.85   412.2 1579.65   441.9 1577.28   491.7 1576.43   560.9 1565.33
   561.3 1565.28   571.3 1565.58   575.9 1566.94   581.2 1568.51   611.1 1583.36
   640.9 1594.61   650.9  1596.5   680.7 1596.14   690.7 1598.82   800.1 1657.34
   879.7 1704.04   959.3 1747.18   969.3 1749.27   999.1 1751.64  1038.9 1747.18
#Mann= 3 , 0 , 0
       0      .1       0   560.9    .045       0   575.9      .1       0
Bank Sta=560.9,575.9
XS Rating Curve= 0 ,0
Exp/Cntr=0.3,0.1

Type RM Length L Ch R = 1 ,6658.3  ,292,297.9,303.8
XS GIS Cut Line= 3
     1964909.877      375753.955     1964660.104      376389.598
     1964117.831      376738.991
#Sta/Elev= 30
       0 1781.21    49.5 1779.23    89.1  1779.1   178.2 1774.98     198  1771.9
   207.9 1769.45   237.6 1759.63   356.3 1717.83   494.9 1670.82   534.5 1655.67
     584 1637.96   643.4  1614.4     683 1600.61   722.6 1583.59   772.3 1563.99
   782.2  1561.1   817.5 1553.53   831.8  1552.4   832.5 1552.52   881.4 1563.48
     941 1572.64   980.7 1583.13  1000.5 1586.93  1010.5 1587.57  1020.4 1587.16
  1040.2 1582.73  1050.2 1583.25  1060.1 1587.16  1248.6 1679.06    1328 1714.06
#Mann= 3 , 0 , 0
       0      .1       0   817.5    .045       0   832.5      .1       0
Bank Sta=817.5,832.5
XS Rating Curve= 0 ,0
Exp/Cntr=0.3,0.1

Type RM Length L Ch R = 1 ,6360.4  ,295.9,297.8,299.7
XS GIS Cut Line= 3
     1964859.645      375698.947     1964495.847      376183.258
     1963886.945      376379.725
#Sta/Elev= 30
       0 1785.61    99.3 1772.02   119.2 1767.94   268.1 1704.18   377.3 1660.67
   466.7 1628.59   556.1 1601.23   605.7 1589.34   625.7 1580.61   675.7 1551.82
   705.7 1540.36   721.1 1537.83   725.7 1537.64   736.1 1538.35   785.7 1543.12
   845.7 1564.12   875.6 1577.63   905.6 1593.28   945.6 1616.81   965.6  1630.2
   995.6 1653.77  1005.6 1660.36  1125.6 1724.87  1145.6 1734.24  1155.6 1736.56
  1185.6 1738.35  1195.6 1741.82  1205.6 1747.75  1215.6 1755.72  1245.5 1784.29
#Mann= 3 , 0 , 0
       0      .1       0   721.1    .045       0   736.1      .1       0
Bank Sta=721.1,736.1
XS Rating Curve= 0 ,0
Exp/Cntr=0.3,0.1

Type RM Length L Ch R = 1 ,6062.6  ,294,292.9,286.6
XS GIS Cut Line= 3
     1964835.986      375632.504     1964439.616      375909.923
      1963824.48      376052.851
#Sta/Elev= 30
       0 1785.24    49.4 1778.11      79 1771.22    98.7 1764.31   286.3  1662.6
   385.1 1610.85   473.9 1555.96   493.7 1545.99   533.2  1530.1     543  1527.1
   548.9 1526.67   552.9 1526.38   563.9 1527.35   602.2 1533.83   651.6 1544.75
   700.9 1557.19   720.6 1564.49   740.4 1573.84     770 1591.13   819.3  1623.1
     918 1684.18   977.2 1725.14   996.9 1736.61  1016.7  1744.4  1026.5  1745.2
  1036.4 1743.06    1066 1732.05  1075.9 1732.71  1085.7  1739.5  1115.3 1767.73
#Mann= 3 , 0 , 0
       0      .1       0   548.9    .045       0   563.9      .1       0
Bank Sta=548.9,563.9
XS Rating Curve= 0 ,0
Exp/Cntr=0.3,0.1

Type RM Length L Ch R = 1 ,5769.5  ,348.9,343,342.4
XS GIS Cut Line= 3
     1964783.202      375508.864     1964256.588      375657.026
     1963773.309       375926.46
#Sta/Elev= 30
       0 1775.55    39.8 1771.05    49.7 1768.29    59.7 1762.91   288.4 1623.91
   328.2 1597.42   338.2 1591.74   348.1 1587.87   397.9 1575.18   427.7 1565.74
   447.6 1557.04   477.4 1541.97   527.2 1518.78   537.1  1514.6   539.6 1514.31
   547.1 1513.44   554.6 1514.74   645.9 1544.31   665.6 1552.11   744.7 1596.73
   843.5 1654.91   912.6 1692.83   952.2 1716.74   991.7  1742.1  1001.6 1745.56
  1011.4 1745.54  1031.2 1741.24  1080.6 1726.62  1090.5  1725.9  1100.4 1729.87
#Mann= 3 , 0 , 0
       0      .1       0   539.6    .045       0   554.6      .1       0
Bank Sta=539.6,554.6
XS Rating Curve= 0 ,0
Exp/Cntr=0.3,0.1
